--- JACKSBR.prj (project) ---

Proj Title=JACKSBR
Current Plan=p01
Default Exp/Contr=0,0
English Units
Geom File=g01
Flow File=f01
Plan File=p01
BEGIN DESCRIPTION:
END DESCRIPTION:
DSS Export Rating Curves= 0
DSS Export Rating Curve Sorted= 0
DSS Export Volume Flow Curves= 0
DXF OffsetX= 0
DXF OffsetY= 0
DXF ScaleX= 0
DXF ScaleY= 0

--- JACKSBR.p01 (plan) ---

Plan Title=Floodplain
Program Version=4.00
Geom File=g01
Flow File=f01
K Sum by GR=0
Std Step Tol=0.01
Critical Tol=0.01
Num of Std Step Trials=20
Max Error Tol=0.3
Flow Tol Ratio=0.001
Split Flow NTrial=30
Split Flow Tol=0.02
Split Flow Ratio=0.02
Log Output Level=0
Friction Slope Method=1
Unsteady Friction Slope Method=2
Unsteady Bridges Friction Slope Method=1
Global Log Level=0
CheckData=False
Run HTab=0
Run UNet=0
Run PostProcess=0
UNET Theta=0
UNET Theta Warmup=0
UNET ZTol=0
UNET ZSATol=0
UNET MxIter=0
UNET MaxInSteps=0
UNET DtIC=0
UNET DtMin=0
UNET MaxCRTS=0
UNET WFStab=0
UNET SFStab=0
UNET WFX=0
UNET SFX=0
UNET DSS MLevel=0
UNET DZMax Abort=0
UNET Convert EG Bridges=0
UNET Use Existing IB Tables=0
UNET Froude Limit=0
UNET Froude Power=0
Write IC File=0
Echo Input=False
Echo Output=False
Write Detailed=0

--- JACKSBR.f01 (steady flow) ---

Flow Title=NFF Regression Equation
Program Version=4.00
Number of Profiles=1
Profile Names=P100yr
River Rch & RM=JACKSBR,Main      ,9751.7
889.5818
River Rch & RM=JACKSBR,Main      ,9216.8
928.1571
River Rch & RM=JACKSBR,Main      ,6969
1009.558
River Rch & RM=JACKSBR,Main      ,4966.4
1120.875
River Rch & RM=JACKSBR,Main      ,899.4
1241.739
River Rch & RM=JACKSBR,Main      ,595.3
1244.205
Boundary for River Rch & Prof#=JACKSBR,Main      ,1
Up Type=0
Dn Type=3
Dn Slope=0.004139

--- JACKSBR.g01 (geometry) ---

Geom Title=USGS 10m DEM
Program Version=4.10

River Reach=JACKSBR         ,Main
Reach XY= 30
     1746721.113      359439.463     1746798.034      359512.823
     1746868.546      359503.564     1747107.144      359618.234
      1747274.52      359485.046     1747721.092      359572.651
     1748147.009      359513.535     1748295.866      359552.708
     1748496.004      359658.831     1749362.083      360356.822
     1749399.325      360486.523     1749466.069      360517.645
     1749519.487      360479.184     1749973.181      360819.277
     1750235.404      360916.222     1750442.001      360940.528
     1750634.709      361091.395      1751116.48      360997.646
     1751307.994      361001.108     1751354.327      360936.013
     1751914.691      360824.098     1752319.605      360801.899
     1752629.501        360886.1     1752875.161       361121.17
     1752945.473      361389.399     1752884.862      362119.583
      1753018.39      362428.635     1753336.966      362806.239
     1753421.168      363300.597     1753598.251       363379.59

Type RM Length L Ch R = 1 ,9751.7  ,301.5,294.2,286.6
XS GIS Cut Line= 3
       1746688.5      359496.592     1746729.865      359444.299
      1746776.16      359360.529
#Sta/Elev= 30
       0  944.99     3.9  945.12     7.8  944.92    15.7  944.24    47.1   942.6
      51     941    54.9  938.81    59.2   937.4    62.8  936.65    66.7  936.42
    70.7  936.72    74.2  937.52    78.6  939.15    82.6  940.81    86.6  941.39
    90.6  940.77    94.6  940.42    98.6  940.29  106.19940.3659   110.5  941.09
   114.5  944.31   118.5  948.31   122.5  951.69   126.5  954.21   130.5  956.35
   138.5  960.44   142.4  962.24   146.4  964.29   158.4  971.42   162.4  974.38
#Mann= 4 ,-1 , 0
       0     .12       0    59.2    .045       0    74.2    .016       0
  106.19     .12       0
Bank Sta=59.2,74.2
XS Rating Curve= 0 ,0
Exp/Cntr=0.3,0.1

Type RM Length L Ch R = 1 ,9457.5  ,249.1,240.7,228.7
XS GIS Cut Line= 2
     1746945.829      359642.618     1747013.537      359407.722
#Sta/Elev= 30
       0  964.32     7.9   960.6    15.8  957.28    31.5  946.35    39.4  940.08
    47.3  934.99    51.3  933.46    55.2  932.76      67  932.04    78.9  931.81
    86.7   930.4    90.7  930.21    94.6   930.5   100.3  932.17   110.4  936.01
   114.3  937.04   118.3  937.05   126.2  935.65   130.1  935.32  150.18934.3167
   157.7   934.4   165.6   934.1  180.92934.2664   189.3  934.36   197.1   933.6
   201.1  934.21     205  935.54     209   937.2   232.6  948.95   244.5   958.1
#Mann= 5 ,-1 , 0
       0     .12       0    78.9    .045       0   100.3     .12       0
  150.18    .016       0  180.92     .12       0
Bank Sta=78.9,100.3
XS Rating Curve= 0 ,0
Exp/Cntr=0.3,0.1

Type RM Length L Ch R = 1 ,9216.8  ,78.3,55.7,35.2
XS GIS Cut Line= 3
     1747166.685      359670.366     1747185.349      359593.109
     1747141.512      359406.044
#Sta/Elev= 30
       0  946.67       8  945.09    23.8  940.51    35.8  937.95    51.7  936.51
    59.6  935.16    63.6  933.83    71.5  929.42    75.5  927.73    83.4  926.58
    95.2  926.05    99.1  926.53     103  927.68   106.9   928.1   114.8  927.58
   142.2  927.64  146.52 928.356     154  931.09   157.9  931.67  176.85931.6166
   185.4  931.08   193.2  928.36   197.1  927.86   212.8  932.24   220.6  935.89
   228.5  940.68   236.3  946.36   244.2  955.09     252  962.14   271.6  981.61
#Mann= 5 ,-1 , 0
       0     .12       0    83.4    .045       0    99.1     .12       0
  146.52    .016       0  176.85     .12       0
Bank Sta=83.4,99.1
XS Rating Curve= 0 ,0
Exp/Cntr=0.3,0.1

Type RM Length L Ch R = 1 ,9161.1  ,38.8,51.4,66.7
XS GIS Cut Line= 4
     1747260.869      359642.155     1747242.136      359559.627
     1747195.308      359533.764     1747195.829      359407.722
#Sta/Elev= 30
       0   942.4    26.9   935.8    53.8  931.71    61.6  931.53    73.1  929.73
    88.4  928.72    96.1  927.24   103.8  925.07   111.4  924.68   118.8   925.8
   122.8  926.85   138.1  927.68  144.05 929.975     146   930.6   149.9  930.97
   161.8  931.43   169.6  931.53  173.58930.8036   177.5  928.78   181.4  926.19
   185.4  924.79   189.3  925.57   193.3  927.02   205.1  933.85     213  938.74
   216.9  941.81   232.6  955.58   248.4   970.9   260.2  983.32   264.2  986.78
#Mann= 5 ,-1 , 0
       0     .12       0   103.8    .045       0   118.8     .12       0
  144.05    .016       0  173.58     .12       0
Bank Sta=103.8,118.8
XS Rating Curve= 0 ,0
Exp/Cntr=0.3,0.1

Type RM Length L Ch R = 1 ,9109.7  ,43.3,53.5,60.6
XS GIS Cut Line= 4
      1747283.85      359641.055     1747259.133      359513.682
     1747238.016      359495.743     1747241.141      359409.284
#Sta/Elev= 30
       0  936.86    15.7  934.34    39.3  934.13    47.2  933.73      59   932.5
    62.9  931.94    82.6  927.46   85.25927.2833    94.4  928.12     114  928.47
     118     928   121.9  927.04   129.8  923.49   134.9  921.89   137.7   921.4
   145.6  921.22   149.9  921.53   153.5  922.03   161.4  921.54   165.3  922.19
   169.2  923.78   177.1  927.76     185  933.26   188.9  936.57   216.4  967.34
   220.4  971.69   228.2  979.33   232.2  983.19   236.1  986.22     244   990.7
#Mann= 5 ,-1 , 0
       0     .12       0   85.25    .016       0   134.9    .045       0
   149.9    .016       0   153.5     .12       0
Bank Sta=134.9,149.9
XS Rating Curve= 0 ,0
Exp/Cntr=0.3,0.1

Type RM Length L Ch R = 1 ,9056.2  ,299.5,304.5,302.9
XS GIS Cut Line= 2
     1747309.915      359633.474     1747285.175      359403.873
#Sta/Elev= 30
       0   936.9    11.9  939.99    23.9  939.32    35.8  935.95    39.8  934.34
    47.8  930.17    59.7  927.81    67.7   924.2    71.7   924.1   76.55925.3793
    79.6  926.34  106.25927.8694   107.5  927.91   115.5  925.35   119.4  924.77
   135.4  923.87   142.5  921.11   151.3  920.49   157.5  921.01   159.3   921.4
   163.2  924.14   171.2  932.63   183.2  943.96   191.1  952.03   195.1  957.25
   199.1  963.75   203.1  969.15     215  981.67     223  988.35   230.9  993.03
#Mann= 5 ,-1 , 0
       0     .12       0   76.55    .016       0  106.25     .12       0
   142.5    .045       0   157.5     .12       0
#XS Ineff= 2 , 0
          107.74  928.59
Permanent Ineff=
       F       F
Bank Sta=142.5,157.5
XS Rating Curve= 0 ,0
Exp/Cntr=0.3,0.1

Type RM Length L Ch R = 1 ,8751.7  ,277.5,273.4,275.3
XS GIS Cut Line= 3
     1747572.815      359643.985     1747582.818      359535.768
     1747570.287       359464.86
#Sta/Elev= 30
       0  920.97     7.8  921.13    15.5  921.06    23.3  921.35      31   920.9
    38.8  921.03    42.7  920.78    46.6  919.84    50.5  918.65    54.3  917.94
   57.33918.2508      66  918.61    73.8  919.25    77.6  918.72    81.5  917.47
    85.4  915.76      87915.3661    89.3   914.8    93.2  914.14      97  913.38
   100.9  913.22   108.7  913.65   112.5  914.26   123.8  916.38   131.4   918.3
     139  919.77   146.6  921.72   150.4  922.43   161.7     923   180.7  927.83
#Mann= 5 ,-1 , 0
       0     .12       0   57.33    .016       0      87     .12       0
    93.2    .045       0   112.5     .12       0
#XS Ineff= 2 , 0
           73.48  919.43
Permanent Ineff=
       F       F
Bank Sta=93.2,112.5
XS Rating Curve= 0 ,0
Exp/Cntr=0.3,0.1

Type RM Length L Ch R = 1 ,8478.3  ,197.3,198.6,199.8
XS GIS Cut Line= 2
     1747847.426      359637.861     1747831.801      359446.889
#Sta/Elev= 30
       0  944.12       4   940.4       8  937.48      16  933.35   21.51929.8192
      24  928.07    31.9  920.67    35.9   917.9    39.9  917.05   51.15916.3244
    55.9  914.63    63.2  909.77    63.9  909.33    67.9  909.04    75.8  909.37
    78.2  910.06    83.8  912.29    99.8  920.48   107.8  923.14   111.8  923.98
   115.8  923.85   123.8   921.9   131.7  918.92   135.7  918.12   139.7   918.6
   163.7  928.11  169.68  929.29   175.6  929.95   183.6  929.44   191.6  929.58
#Mann= 6 ,-1 , 0
       0     .12       0   21.51    .016       0   51.15     .12       0
    63.2    .045       0    78.2     .12       0  169.68      .1       0
Bank Sta=63.2,78.2
XS Rating Curve= 0 ,0
Exp/Cntr=0.3,0.1

Type RM Length L Ch R = 1 ,8279.7  ,76.7,70.3,66.7
XS GIS Cut Line= 2
     1748038.763      359620.103     1748033.121      359403.089
#Sta/Elev= 30
       0  932.81       4  931.11    11.8  929.77    15.8  927.75    23.7  921.98
   33.24913.9199    35.5  911.88    39.5  909.28    43.4  908.04    47.4  907.54
    51.3  907.55   62.78908.1458    67.1  908.26      75  907.32    82.9  906.32
    90.8  906.64    94.7  907.27   106.6   911.3   110.5  911.47   118.4  909.39
   122.4   909.5   130.2  913.57   134.2  914.38   142.1   914.6   153.9  916.55
   181.6  918.48   185.5  919.34   197.4  924.24   209.2  930.37   217.1  932.66
#Mann= 5 ,-1 , 0
       0     .12       0   33.24    .016       0   62.78     .12       0
      75    .045       0    94.7      .1       0
Bank Sta=75,94.7
XS Rating Curve= 0 ,0
Exp/Cntr=0.3,0.1

Type RM Length L Ch R = 1 ,8209.4  ,28,27.9,22.6
XS GIS Cut Line= 4
     1748090.296        359628.7      1748115.47      359531.478
     1748097.458      359509.598     1748132.079      359415.676
#Sta/Elev= 30
       0  933.07    23.2  918.94      27  917.62    30.9  917.04    34.8  915.44
    46.4  909.03    50.2  907.56    54.1  906.77    65.7  905.81   73.71 906.145
      85  906.81    96.6  908.38   100.4  908.37  105.19907.8122   108.2  907.34
   121.7  905.99   125.2  907.65   128.8  909.24   132.6  910.44   136.5   911.1
   151.9  911.64   167.3  910.29   171.1  910.51     175  911.26   178.8   912.6
   182.7  914.32   190.4  918.42   198.1  923.09   217.3   935.9   228.9   945.2
#Mann= 5 ,-1 , 0
       0     .12       0   73.71    .016       0  105.19      .1       0
   108.2    .045       0   125.2      .1       0
Bank Sta=108.2,125.2
XS Rating Curve= 0 ,0
Exp/Cntr=0.3,0.1

Type RM Length L Ch R = 1 ,8181.5  ,67.6,79.9,94.6
XS GIS Cut Line= 4
     1748115.152       359634.86      1748142.93      359527.655
     1748121.662      359500.745      1748151.61      359420.884
#Sta/Elev= 30
       0   932.7    11.9  925.92    27.7  918.74    35.6  913.54    51.4  908.63
    63.3  905.98    67.2  905.35   80.08905.7516      91  906.41   102.8  907.74
  110.59908.1063   114.6  907.82   118.4  907.12   122.2  905.65   129.8  904.23
   133.6   904.1   137.4  905.51   141.2  908.98     145  910.31   152.8   910.9
   160.6  910.38   164.4   910.7   172.2  912.84   176.1  914.45   183.8  916.62
   187.7  918.05   199.3  924.62   203.2  927.39     211  933.71   230.3  945.99
#Mann= 5 ,-1 , 0
       0     .12       0   80.08    .016       0  110.59      .1       0
   122.2    .045       0   137.4      .1       0
#XS Ineff= 2 , 0
       0  110.59  908.11               0
Permanent Ineff=
       F       F
Bank Sta=122.2,137.4
XS Rating Curve= 0 ,0
Exp/Cntr=0.3,0.1

Type RM Length L Ch R = 1 ,8101.6  ,343.3,349.8,356
XS GIS Cut Line= 2
      1748185.03       359641.37     1748232.339      359438.245
#Sta/Elev= 30
       0  921.72    15.7  912.76    27.6  907.32    31.5  906.35    47.2  906.68
   55.96905.9179      63  904.67    66.9  903.73    70.8  903.31    78.7  904.16
   86.28904.3288    98.4  905.61   102.3  905.24   110.2   901.2   111.8  900.75
   114.1   900.1     118  899.59     122  900.06   125.9  901.33   133.8  904.78
   137.7  906.92   141.7  910.17   157.4   925.4   161.3  928.76   165.3  931.45
   169.2  933.07  177.26935.2116   188.9  937.48   200.7  940.61   208.6  942.37
#Mann= 6 ,-1 , 0
       0     .12       0   55.96    .016       0   86.28      .1       0
   111.8    .045       0   125.9      .1       0  177.26     .12       0
#XS Ineff= 2 , 0
       0    98.4  905.61               0
Permanent Ineff=
       F       F
Bank Sta=111.8,125.9
XS Rating Curve= 0 ,0
Exp/Cntr=0.3,0.1

Type RM Length L Ch R = 1 ,7751.8  ,248.9,253.4,257.9
XS GIS Cut Line= 2
     1748462.634      359786.205     1748552.912      359625.788
#Sta/Elev= 30
       0  927.77     3.9  924.69    11.8  915.92    15.7  912.22    19.6  909.37
    27.4  904.56    31.3  900.97    35.2  898.64   36.89897.9302    39.2  896.96
    43.1  896.43    54.8  896.39   59.28896.0933    66.6  895.35    70.5  895.37
    78.3  896.03   97.11896.4404   101.8  895.53   109.7  892.79   112.8     892
   117.5  891.71   127.8  892.04   129.2   892.2   133.2  894.49   137.1  897.46
   152.7  904.57   164.5  911.53   172.3  916.66   176.2  918.49   184.1  921.44
#Mann= 6 ,-1 , 0
       0     .12       0   36.89      .1       0   59.28    .016       0
   97.11      .1       0   112.8    .045       0   127.8      .1       0
#XS Ineff= 2 , 0
       0   94.42                       0
Permanent Ineff=
       F       F
Bank Sta=112.8,127.8
XS Rating Curve= 0 ,0
Exp/Cntr=0.3,0.1

Type RM Length L Ch R = 1 ,7498.3  ,244.7,246.6,248.7
XS GIS Cut Line= 2
      1748649.51      359917.375     1748772.773      359775.014
#Sta/Elev= 30
       0   924.8     7.8  918.59   12.89914.9225    27.5  904.89    31.4  901.65
    39.2  894.58    43.2  893.01      51   891.5   58.01 891.138    70.6  892.41
    86.3  892.65    90.2  892.26    98.1   890.5  103.13 888.194   103.9  887.89
   105.9   887.1   109.8  886.54   113.8   886.9   117.7   888.3   121.6   890.7
   129.5  898.83   133.4  902.43   137.3  905.62   141.2   908.4  148.25912.3219
     153  914.54   160.8  917.48   168.7   920.8   172.6  921.81   188.3  924.25
#Mann= 7 ,-1 , 0
       0     .12       0   12.89      .1       0   58.01    .016       0
  103.13      .1       0   103.9    .045       0   117.7      .1       0
  148.25     .12       0
#XS Ineff= 2 , 0
       0   82.27                       0
Permanent Ineff=
       F       F
Bank Sta=103.9,117.7
XS Rating Curve= 0 ,0
Exp/Cntr=0.3,0.1

Type RM Length L Ch R = 1 ,7251.7  ,284.3,282.6,281
XS GIS Cut Line= 3
     1748818.222      360082.823     1748898.189      360005.875
     1748942.978      359962.777
#Sta/Elev= 30
       0  919.61       4  916.34     7.9  912.73    11.9  909.35    15.8  906.92
    27.7  900.08    31.7  898.16    43.6   893.2    51.5  889.05    59.4  886.49
    64.5885.4407    67.4   885.1    79.3  886.45    91.2  886.62    95.1   886.4
    99.1   885.5     103  884.31     107  883.78     111  883.75   114.9  884.12
  118.95885.5981   122.6  888.23   126.5  891.51     142  901.32   145.9  904.11
   149.8  907.13   153.7   909.6   157.6  911.71   161.5  913.52   173.1  914.82
#Mann= 5 ,-1 , 0
       0      .1       0    64.5    .016       0     103    .045       0
   114.9      .1       0  118.95     .12       0
Bank Sta=103,114.9
XS Rating Curve= 0 ,0
Exp/Cntr=0.3,0.1

Type RM Length L Ch R = 1 ,6969    ,215.8,217.4,216.9
XS GIS Cut Line= 2
     1749057.496      360243.764     1749156.454      360132.652
#Sta/Elev= 30
       0  914.09    9.56906.9664    11.8  905.32    15.7  902.83    23.5  898.09
    27.4  896.12    39.2  890.72      47  886.18   49.11885.2115    50.9  884.39
    54.8  884.11    58.7  884.42    62.6  884.45    66.6  884.36    70.5  884.01
    82.1  882.04    86.1  881.46    90.1  880.69      94  880.83    97.9  881.46
   101.8  882.66   105.7  885.49  109.81888.7755   113.6   891.4   125.3  900.72
   129.2  903.33   133.1  906.42     137   910.1     141  913.52   148.8  918.28
#Mann= 6 ,-1 , 0
       0     .06       0    9.56     .05       0   49.11    .016       0
    82.1    .045       0   101.8      .1       0  109.81     .12       0
Bank Sta=82.1,101.8
XS Rating Curve= 0 ,0
Exp/Cntr=0.3,0.1

Type RM Length L Ch R = 1 ,6751.7  ,87.7,89.5,94.3
XS GIS Cut Line= 3
      1749216.99      360378.162     1749289.691      360305.915
     1749337.104      360251.331
#Sta/Elev= 30
       0  893.97    3.03893.1076     3.9  892.86    19.7  892.62    33.2 893.309
    35.5  893.24    39.4  891.66   44.67888.1973    51.2  883.68    55.2  881.68
    59.1  881.73    63.1   882.7      67  882.95    82.8  883.53   86.31 883.062
      95  880.12    98.6  879.07   102.5  878.48   113.9   878.9   117.7  879.96
   121.5  881.83   125.3   884.4   129.1  887.44   136.7  895.07   140.6  898.52
   144.4  901.26     152  905.58   155.8  907.33     171  912.59   174.8  915.28
#Mann= 7 ,-1 , 0
       0      .1       0    3.03     .05       0    33.2      .1       0
   44.67    .016       0   86.31     .12       0      95    .045       0
   117.7     .12       0
#XS Ineff= 2 , 0
       0      67                       0
Permanent Ineff=
       F       F
Bank Sta=95,117.7
XS Rating Curve= 0 ,0
Exp/Cntr=0.3,0.1

Type RM Length L Ch R = 1 ,6662.2  ,71.6,78.2,74.5
XS GIS Cut Line= 4
     1749258.699      360472.924     1749353.317       360358.34
     1749371.112      360357.038     1749401.928      360315.806
#Sta/Elev= 30
       0  902.19     3.9   900.2     7.8  897.35    11.7   893.3    15.6  889.78
    19.6  887.78    23.5   887.6    35.2  888.42    39.1  889.28      43  889.74
    62.6  887.84   76.64 886.902   101.7  885.23   109.5  884.33  114.94884.1153
   125.1  884.57     133  885.51   136.9  884.76   148.6   879.2   149.9   878.8
   155.7  877.36   159.3   877.1   162.9  877.51   166.4  878.73   170.4  880.28
   174.4   882.7   182.3   886.9   194.2  893.98   202.1  896.17   217.9  901.48
#Mann= 5 ,-1 , 0
       0      .1       0   76.64     .06       0  114.94    .016       0
   149.9    .045       0   166.4     .12       0
Bank Sta=149.9,166.4
XS Rating Curve= 0 ,0
Exp/Cntr=0.3,0.1

Type RM Length L Ch R = 1 ,6584    ,60.7,49.7,47.2
XS GIS Cut Line= 4
     1749288.489      360513.201     1749348.109      360435.597
     1749367.206      360436.031     1749430.574       360356.17
#Sta/Elev= 30
       0  917.27     3.9  914.03     7.8  910.35    11.7  907.44    19.6  903.06
    31.3  897.03    35.2  894.24    43.1  887.54    50.9  880.33    54.8  878.22
    66.6  877.62    80.1877.7808   88.07877.7002      90  877.72    97.9  877.67
   101.7  877.36   109.3   877.9     117  879.26   120.9  881.12   124.8  882.29
   132.6  883.93   152.2  885.06   160.1  886.19  163.86886.1225   179.7  885.27
   183.6   886.5   195.4  888.81   211.1  893.15     215  893.73   218.9   894.7
#Mann= 6 ,-1 , 0
       0      .1       0    80.1     .04       0   88.07     .06       0
      90     .04       0     117    .016       0  163.86     .12       0
Bank Sta=97.9,117
XS Rating Curve= 0 ,0
Exp/Cntr=0.3,0.1

Type RM Length L Ch R = 1 ,6534.3  ,50.1,50.1,50.1
XS GIS Cut Line= 2
     1749354.446      360525.488     1749441.251      360396.582
#Sta/Elev= 30
       0  904.42       4  903.63       8  902.64      12  900.35    15.9  897.39
    19.9  893.72    23.9  889.85   27.79886.5629    35.9  879.79    39.8  878.24
    43.8  877.97    47.8  877.94    55.8  877.42    59.8  877.44    63.8  877.62
    75.7  878.51    79.7  878.99    83.7  880.18    91.6  882.68    95.6  883.59
    99.6  883.79   103.6  884.11   111.6   884.6   119.6  885.42   123.5  885.52
  127.91  885.24   139.5  885.39   143.4  885.95   151.4  888.01   155.4  888.75
#Mann= 5 ,-1 , 0
       0      .1       0   27.79     .04       0    39.8     .04       0
    75.7    .016       0  127.91     .12       0
Bank Sta=39.8,75.7
XS Rating Curve= 0 ,0
Exp/Cntr=0.3,0.1

Type RM Length L Ch R = 1 ,6484.2  ,48.7,44.1,57.6
XS GIS Cut Line= 2
     1749396.067      360552.932     1749482.872      360424.026
#Sta/Elev= 30
       0  910.12       8  905.78    15.9  901.12    19.9  898.47    23.9   895.1
   25.27893.7368    31.9  887.04    35.9  882.71    39.8  879.17    43.8  878.03
    51.8  877.46    59.8   877.3    67.7  877.32    71.7  877.65    75.7  878.99
    79.7  880.78    83.7  881.84    87.7   882.7    91.6   883.2   96.49883.4045
   103.6  883.63   107.6   883.9   115.6  885.02   119.6  885.45   123.5  884.97
   127.5  883.83   132.1884.3085   135.5  884.64   139.5   885.3   155.4  891.58
#Mann= 6 ,-1 , 0
       0      .1       0   25.27     .04       0    43.8     .04       0
    71.7     .06       0   96.49    .016       0   132.1     .12       0
Bank Sta=43.8,71.7
XS Rating Curve= 0 ,0
Exp/Cntr=0.3,0.1

Type RM Length L Ch R = 1 ,6440.1  ,41.1,59,43.4
XS GIS Cut Line= 4
     1749436.112       360580.48     1749472.675      360520.667
     1749466.165      360511.118      1749513.04      360436.031
#Sta/Elev= 30
       0  909.99    11.7  902.58    15.6  899.64    23.4  891.46    31.2  883.76
      35   880.6   37.05879.3136      39  878.09    42.8   877.3   56.86877.0397
    58.4  877.02    62.3  877.02    66.2   877.5    70.1  878.53      74  878.51
    77.8  878.87    81.7  879.01    91.9 881.559      97  882.28   120.2     884
  126.72883.9771   131.7  884.04   139.4  883.71   143.2   884.2   147.1  885.06
   150.9   885.5   154.8  886.76   162.5  891.82   166.3  893.74   170.2  895.32
#Mann= 7 ,-1 , 0
       0      .1       0   37.05     .04       0   56.86      .1       0
    58.4     .04       0    77.8      .1       0    91.9    .016       0
  126.72     .12       0
Bank Sta=70.1,81.7
XS Rating Curve= 0 ,0
Exp/Cntr=0.3,0.1

Type RM Length L Ch R = 1 ,6381.1  ,91,80.7,83.6
XS GIS Cut Line= 4
     1749454.931      360587.697     1749520.505      360485.771
     1749513.908       360476.83     1749536.477      360442.108
#Sta/Elev= 30
       0  907.14     7.8  902.33    11.7   899.4    19.6  891.42    23.5  888.27
   31.15883.0069    35.2  881.42    39.1  880.99      43  881.07   55.52882.4136
   66.27883.0688    74.3  881.63    78.2   881.3    97.7  882.34   101.6  881.77
   105.6  880.38   110.1  877.62   117.3  872.13   121.2  870.26   124.9  869.92
   136.1  870.46   139.8  872.17   143.6   875.4   151.1  880.61   154.9  883.98
   158.7   888.2   162.4  891.84   166.2  894.17  172.23896.9765   173.7  897.64
#Mann= 8 ,-1 , 0
       0      .1       0   31.15     .04       0   55.52      .1       0
   66.27    .016       0   110.1      .1       0   121.2    .045       0
   136.1      .1       0  172.23     .12       0
Bank Sta=121.2,136.1
XS Rating Curve= 0 ,0
Exp/Cntr=0.3,0.1

Type RM Length L Ch R = 1 ,6300.4  ,228.3,228.8,229.2
XS GIS Cut Line= 2
     1749519.463      360621.361     1749608.021      360484.859
#Sta/Elev= 30
       0  905.56     7.9  900.34    11.9  896.88    19.8   888.6    23.8  886.08
    31.8  882.84    47.6  878.34    51.6   877.6    59.5  877.77    67.5  878.78
   71.35878.9083    79.4  879.03    87.3  879.53    91.3   879.1    95.2  876.94
   103.2  868.24   105.3  867.34   107.2  866.52   111.1  866.45   115.1  866.53
   119.1  867.32   120.3  867.96     123   869.4     127  872.62   134.9  880.16
  141.77885.5953   146.8  888.91   150.8  890.95   158.7  894.29   162.7  896.42
#Mann= 5 ,-1 , 0
       0      .1       0   71.35    .016       0   105.3    .045       0
   120.3      .1       0  141.77     .12       0
Bank Sta=105.3,120.3
XS Rating Curve= 0 ,0
Exp/Cntr=0.3,0.1

Type RM Length L Ch R = 1 ,6071.6  ,376.9,374,371.1
XS GIS Cut Line= 3
     1749727.685      360721.088     1749759.116       360670.65
     1749796.563      360615.241
#Sta/Elev= 30
       0  883.02       4  880.15     7.9  876.72    11.9  873.66   14.04872.4089
    15.8  871.38    19.8  869.52    23.8  869.02    31.7  869.51    39.6   869.8
    43.6   870.1    47.5  870.18   48.84870.0359    51.5  869.75    59.4  867.87
    63.4  866.68    71.2  864.56    79.1  861.89      83  861.19      87  861.36
    92.1  862.22    94.8  862.64   97.32864.1394    98.8  865.02   102.7  868.56
   106.6  872.41   114.5  879.54   118.4  883.36   122.4  887.84   126.3  891.29
#Mann= 6 ,-1 , 0
       0      .1       0   14.04    .016       0   48.84      .1       0
    79.1    .045       0    92.1      .1       0   97.32     .12       0
Bank Sta=79.1,92.1
XS Rating Curve= 0 ,0
Exp/Cntr=0.3,0.1

Type RM Length L Ch R = 1 ,5697.6  ,227.6,221.8,216
XS GIS Cut Line= 2
     1750016.685      360965.806     1750113.908      360775.528
#Sta/Elev= 30
       0  874.95     7.9  873.42    11.9  872.44    15.8  871.35   22.86868.6423
    27.7  866.95    31.7  866.28    39.6  866.61    51.4  866.75   64.78867.2834
    67.3  867.17    75.2  864.44      87  858.74    89.2858.1515      91  857.67
   106.8  856.24   110.8  856.21   122.7  856.66   134.5     856   146.4  855.37
   154.3  856.19   162.2  857.66   170.2  859.66     182  861.09     186  862.03
   189.9  863.23   193.9  864.68   197.8  866.62   201.8  868.86   213.7  876.23
#Mann= 6 ,-1 , 0
       0      .1       0   22.86    .016       0   64.78      .1       0
    89.2     .12       0   134.5    .045       0   154.3     .12       0
Bank Sta=134.5,154.3
XS Rating Curve= 0 ,0
Exp/Cntr=0.3,0.1

Type RM Length L Ch R = 1 ,5475.8  ,214.7,224.1,239.5
XS GIS Cut Line= 2
     1750259.741      361032.472     1750301.408      360842.889
#Sta/Elev= 30
       0  866.99       4   867.4     7.9  867.32    11.9  866.22    15.8  864.64
    19.8  863.48    23.8  862.98    35.6  862.32    43.6  862.06   58.87862.0859
    71.3  861.69    79.2  861.69    83.2  860.64    91.1  856.62      99  853.14
     103  852.03   110.9  852.08   118.8  851.88   122.8  852.72   126.8  854.34
   134.7  857.97   138.6  859.47   146.6  861.97   158.5   864.8   162.4   865.9
   166.4  867.68   178.3  875.25   182.2  878.11   186.2  880.76   194.1  885.13
#Mann= 4 ,-1 , 0
       0      .1       0   58.87     .12       0     103    .045       0
   118.8     .12       0
Bank Sta=103,118.8
XS Rating Curve= 0 ,0
Exp/Cntr=0.3,0.1

Type RM Length L Ch R = 1 ,5251.7  ,50.7,59.1,58.8
XS GIS Cut Line= 3
      1750423.63      361070.974     1750487.132      360983.669
     1750540.399      360940.639
#Sta/Elev= 30
       0     859       4  859.23    9.15859.1782      32  858.49      40  858.55
   45.67858.3582      64  857.86      68  857.95      72  857.86      76  856.97
      80  855.39   82.19854.1417      84  853.11      88  851.39      92  850.22
     100  848.94     104  848.64     108  848.57   115.5  848.74  116.75  849.05
   119.4  849.79   123.2   851.5   130.8  855.73   134.6  857.24   153.6  860.52
   161.2  863.28     165  864.33   168.8  865.06   172.6  865.48   176.4  865.57
#Mann= 6 ,-1 , 0
       0      .1       0    9.15    .016       0   45.67      .1       0
   82.19     .12       0     100    .045       0  116.75     .12       0
Bank Sta=100,116.75
XS Rating Curve= 0 ,0
Exp/Cntr=0.3,0.1

Type RM Length L Ch R = 1 ,5192.6  ,55.7,65.2,70.7
XS GIS Cut Line= 4
     1750493.074      361113.722     1750507.658      361034.556
     1750540.296      361022.056     1750570.158      360951.222
#Sta/Elev= 30
       0  872.48     3.8  868.94    11.5  863.42    15.3  861.11   20.96858.6417
    26.8  856.15    34.5  854.11    38.3  854.11   50.99 855.816    57.5  856.26
      69  855.57    80.5  852.85   81.95852.1844    88.3  849.46    92.2  848.79
    99.9  848.56   103.8  849.07   111.6  851.53   119.3  855.17     127   855.1
   134.5855.9954   142.4  856.41   146.2  857.11     150  858.66   153.9  859.39
   165.4  859.92   173.1  859.55   180.8  859.69   188.5  860.41   192.3  861.59
#Mann= 7 ,-1 , 0
       0     .12       0   20.96      .1       0   50.99    .016       0
   81.95      .1       0    88.3    .045       0   103.8      .1       0
   134.5     .12       0
Bank Sta=88.3,103.8
XS Rating Curve= 0 ,0
Exp/Cntr=0.3,0.1

Type RM Length L Ch R = 1 ,5127.4  ,192.1,161,136.4
XS GIS Cut Line= 4
     1750533.352      361146.361     1750546.546      361074.139
     1750601.408       361060.25     1750611.824      360958.861
#Sta/Elev= 30
       0   890.3     3.9  888.45    11.6  881.88   24.11 873.246    38.6  863.01
    46.4  857.09   54.13852.2874      58  850.67    61.8  850.07    73.4  850.07
      81   848.8    88.5  846.87    92.3   846.9      96   848.1    99.4  848.66
   103.6  847.87   107.4  846.34   111.2  845.38   118.7  846.65   126.2  848.74
     130  849.38   137.8  851.91   145.7  852.96   173.1  852.72  186.05853.9363
   204.5  856.44  215.75857.0523   224.1   858.2     228  859.33   231.9  861.43
#Mann= 7 ,-1 , 0
       0      .1       0   24.11     .12       0   54.13      .1       0
    99.4    .045       0   126.2    .016       0  186.05      .1       0
  215.75     .12       0
#XS Ineff= 2 , 0
       0    73.4                       0
Permanent Ineff=
       F       F
Bank Sta=99.4,126.2
XS Rating Curve= 0 ,0
Exp/Cntr=0.3,0.1

Type RM Length L Ch R = 1 ,4966.4  ,314.1,308.7,302.7
XS GIS Cut Line= 2
     1750729.185      361172.537      1750736.13      360969.412
#Sta/Elev= 30
       0  892.72       4  889.33       8  886.61    27.9  875.72    39.8  867.06
    47.8  861.81    63.8  849.14    67.8  846.81    71.7  845.32    75.7  844.51
    87.7  843.55    95.6  842.21    99.6  842.21   103.6  843.28  109.03 845.705
   115.6  849.13   119.6  850.41   123.5   850.7   131.5  850.47  138.59851.7917
   143.5  851.53   151.4  849.97   155.4  849.56  168.14848.9404   175.4  848.63
   179.3  848.88   183.3  850.68   191.3   856.1  197.69859.1832   203.2  862.18
#Mann= 7 ,-1 , 0
       0     .12       0    87.7    .045       0   103.6     .12       0
  109.03      .1       0  138.59    .016       0  168.14     .06       0
  197.69     .12       0
Bank Sta=87.7,103.6
XS Rating Curve= 0 ,0
Exp/Cntr=0.3,0.1

Type RM Length L Ch R = 1 ,4657.7  ,411.6,406,405.8
XS GIS Cut Line= 2
     1751047.079      361099.666     1751007.148      360917.375
#Sta/Elev= 30
       0  866.58    11.9  861.98    27.8  857.14    35.7  854.43    51.6  850.12
    63.5  847.17    67.5   844.9    71.5  842.17    75.4  839.84    79.4   837.9
    80.5  837.67    83.4  837.08    87.4  836.86    91.3  836.87    95.5  837.56
   97.44838.2952   107.2  841.51   119.1  842.78   123.1  844.34  127.67845.6149
     131  845.76   150.9  844.52   154.8  844.54  157.91845.3719   158.8  845.61
   162.8   848.7   170.7  858.28   174.7  861.87   182.6  868.25   186.6  870.96
#Mann= 6 ,-1 , 0
       0     .12       0    80.5    .045       0    95.5     .12       0
   97.44      .1       0  127.67    .016       0  157.91      .1       0
Bank Sta=80.5,95.5
XS Rating Curve= 0 ,0
Exp/Cntr=0.3,0.1

Type RM Length L Ch R = 1 ,4251.7  ,494,500,499.4
XS GIS Cut Line= 3
     1751427.874      361002.746      1751391.76      360927.743
     1751377.482      360863.118
#Sta/Elev= 30
       0  867.69       4  864.74     7.9  861.56    11.9  857.91    15.9  854.71
    19.8  851.78    27.8  846.04    35.7  841.17    39.6  839.01    43.6  837.22
    51.5   834.2    55.5  832.92    59.5  831.86   63.65831.0581    71.4  829.85
    75.7  829.38    87.1  828.59      91  829.24    94.9  831.34   95.41831.7375
   102.7  837.38   106.6  839.17   110.5  839.28   114.4   838.5   118.3     838
  125.66837.5637   133.9   837.4   137.8  837.77   141.6  838.52   149.4  839.22
#Mann= 6 ,-1 , 0
       0     .12       0   63.65      .1       0    75.7    .045       0
      91      .1       0   95.41    .016       0  125.66     .06       0
Bank Sta=75.7,91
XS Rating Curve= 0 ,0
Exp/Cntr=0.3,0.1

Type RM Length L Ch R = 1 ,3751.7  ,491.1,500,509.1
XS GIS Cut Line= 3
     1751890.958      360890.457     1751878.578      360831.006
     1751850.149      360703.005
#Sta/Elev= 30
       0  831.97     3.8  829.37     7.6  828.76    34.4   828.5    41.8  828.43
    49.3  827.31    53.1  825.29   55.04  822.81    56.9  820.65    60.7  819.32
    64.7  820.64    68.2  823.26    72.6  827.53    76.6  829.14    84.6  827.51
   94.84826.7889   104.4  826.78   112.4  829.52   116.4  831.15  125.09838.3141
   132.2  844.14   140.2  851.71   144.2  854.18   152.1  854.58  155.35855.5306
   160.1  858.47     168  866.82     172  870.25   183.9   878.3   191.8  882.31
#Mann= 7 ,-1 , 0
       0     .12       0    34.4     .05       0   55.04    .045       0
    68.2    .016       0   94.84     .06       0  125.09      .1       0
  155.35     .12       0
#XS Ineff= 2 , 0
       0                    76.2       0
Permanent Ineff=
       F       F
Bank Sta=55.04,68.2
XS Rating Curve= 0 ,0
Exp/Cntr=0.3,0.1

Type RM Length L Ch R = 1 ,3251.7  ,274.3,284.2,293.8
XS GIS Cut Line= 3
     1752360.095      360878.657      1752372.14      360813.414
     1752397.892      360680.436
#Sta/Elev= 30
       0  849.94     3.9  847.36     7.8  844.25    11.7  841.81   22.27833.1446
    31.2  825.95    42.9  818.42    46.8  816.66    50.7  815.42    58.5   811.6
    62.4  810.26    66.4  809.95    78.3  810.44   82.37810.6824    86.3  810.82
   106.2  815.77   110.2  816.45   118.1   816.5   126.1  817.21  142.53817.2034
     150  817.03     158  816.33     162  818.66   169.9  825.78  172.62 826.732
   173.9  827.18   177.9  827.18   181.9   827.8   185.9  829.17   201.8  835.95
#Mann= 7 ,-1 , 0
       0      .1       0   22.27     .12       0    62.4    .045       0
    78.3     .12       0   82.37      .1       0  142.53    .016       0
  172.62      .1       0
Bank Sta=62.4,78.3
XS Rating Curve= 0 ,0
Exp/Cntr=0.3,0.1

Type RM Length L Ch R = 1 ,2967.4  ,227.7,237.1,246.3
XS GIS Cut Line= 2
     1752590.482      360962.514      1752723.63      360775.528
#Sta/Elev= 30
       0  864.98    23.8  848.67    35.6   838.9    47.5  829.71    63.3  818.22
    75.2  808.64    78.2  806.92    83.1  805.09    87.1  805.21      91  806.12
    93.2  807.26    98.9  810.13   102.9  811.66   110.8  815.91   114.8  815.52
   122.7  812.18   126.6  812.65  129.84813.8245   134.6  815.21   138.5  815.02
   146.4  813.18   162.3  811.92   166.1811.9785   170.2  812.65   178.1  812.82
  196.34812.0063  202.36812.0468   217.7  812.58   221.6  813.28   229.6  815.67
#Mann= 7 ,-1 , 0
       0      .1       0    78.2    .045       0    93.2      .1       0
  129.84    .016       0   166.1     .04       0  196.34     .08       0
  202.36     .12       0
Bank Sta=78.2,93.2
XS Rating Curve= 0 ,0
Exp/Cntr=0.3,0.1

Type RM Length L Ch R = 1 ,2730.4  ,340.8,346.6,352.2
XS GIS Cut Line= 2
     1752739.178      361095.792     1752925.792        360982.2
#Sta/Elev= 30
       0  839.05       4  834.89     7.9  831.26    23.8  820.04    31.8  816.24
    47.7  810.17    51.6   807.1    55.6  802.42    57.9  801.74    59.6  801.23
    67.5  800.84    72.9  801.22    99.3  804.91   103.3  805.17   111.2  805.28
   131.1  803.84  132.14804.0747     135  804.72     139  806.46     143  807.14
   154.9  806.04   166.8  806.06   170.8  805.63  175.74805.8964   186.7  806.59
   194.6  806.21   198.6  806.72   201.3807.8203   206.6  810.04   218.5   813.3
#Mann= 6 ,-1 , 0
       0      .1       0    57.9    .045       0    72.9      .1       0
  132.14    .016       0  175.74      .1       0   201.3     .12       0
#XS Ineff= 2 , 0
                          142.02          807.19
Permanent Ineff=
       F       F
Bank Sta=57.9,72.9
XS Rating Curve= 0 ,0
Exp/Cntr=0.3,0.1

Type RM Length L Ch R = 1 ,2383.8  ,346.6,353.5,360.3
XS GIS Cut Line= 2
     1752844.941      361381.478     1753049.802      361317.241
#Sta/Elev= 30
       0  830.17       4   826.3    15.9   815.9    23.9  808.13    27.8  806.01
    35.8  804.19    51.7  799.86    55.7  799.47    63.6  799.32    79.5  798.44
    83.5  797.67    91.4  795.34    95.4  794.89    99.4  794.81   103.4  795.52
   107.4  797.59   111.3  800.35   115.3  802.12   123.2  800.84   139.2  800.03
   151.1  801.05  162.24801.5111     171  802.09  174.37802.9023   174.9  803.03
   178.9  805.34   182.9  809.12   194.8  822.56   198.8  825.57   214.7  834.97
#Mann= 5 ,-1 , 0
       0      .1       0    91.4    .045       0   103.4    .016       0
  162.24      .1       0  174.37     .12       0
#XS Ineff= 2 , 0
                          115.33           802.3
Permanent Ineff=
       F       F
Bank Sta=91.4,103.4
XS Rating Curve= 0 ,0
Exp/Cntr=0.3,0.1

Type RM Length L Ch R = 1 ,2030.3  ,326.9,326.1,325.4
XS GIS Cut Line= 2
     1752849.782       361700.95     1753061.209       361700.95
#Sta/Elev= 30
       0  820.43       8  814.95      12   812.8    27.9  806.31    31.9  804.03
    59.8  791.08    63.8  790.33    71.8  789.83    75.8  790.27    79.8   791.2
    95.7  797.95    99.7  799.45   103.7  800.32   107.7  799.97   119.7  800.54
   123.7  799.42   127.6  797.74   131.6  796.74   143.6  796.68  149.98796.2534
   163.6  795.51  179.51795.1727   183.5  796.24   191.5  796.69   195.5  797.65
   199.5  801.19   203.4  805.89   207.4   809.7  209.05 810.888   211.4  812.58
#Mann= 6 ,-1 , 0
       0      .1       0    59.8    .045       0    79.8      .1       0
  149.98    .016       0  179.51      .1       0  209.05     .12       0
Bank Sta=59.8,79.8
XS Rating Curve= 0 ,0
Exp/Cntr=0.3,0.1

Type RM Length L Ch R = 1 ,1704.2  ,311.1,308.5,305.8
XS GIS Cut Line= 2
     1752826.593       362026.75     1753097.426      362018.069
#Sta/Elev= 30
       0  823.79      12  813.12    23.9  803.64    39.8   788.7    47.2  785.11
    55.8  783.82    62.2  784.71    75.7  790.18    87.7  791.02    95.6  793.68
   103.6  792.58   119.6  795.93  143.71796.9708   155.4   796.4   163.4  791.42
   167.4   789.8  173.26788.9826   195.3  787.44  202.82787.9073   207.2  789.38
   215.2  789.27   219.2  791.07   223.2  791.63  232.37790.7087   235.1  790.62
   239.1  792.64   243.1   799.1     251  810.16     263  822.78     271   829.1
#Mann= 7 ,-1 , 0
       0      .1       0    47.2    .045       0    62.2      .1       0
  143.71     .06       0  173.26    .016       0  202.82      .1       0
  232.37     .12       0
#XS Ineff= 2 , 0
                          151.62          797.48
Permanent Ineff=
       F       F
Bank Sta=47.2,62.2
XS Rating Curve= 0 ,0
Exp/Cntr=0.3,0.1

Type RM Length L Ch R = 1 ,1395.7  ,82.8,83.5,83.2
XS GIS Cut Line= 3
       1752918.7      362307.432     1753153.373      362276.708
     1753218.074      362243.583
#Sta/Elev= 30
       0  791.31    31.6  791.27    35.5  790.65    51.3  783.69    64.9  780.04
   66.04  779.78      75  778.39   83.46   779.8    90.7     784    94.7  784.95
   102.6  783.85   106.5  785.66   114.4  791.84   118.3  792.35   122.3  791.75
  141.35787.5634   153.8  784.48   161.7  783.45   193.3  783.32  200.92782.0369
   205.1  782.25     217  786.91  230.71787.0845   244.3  785.97     252   786.6
   255.8  787.73   259.6   790.1   271.1  800.37   290.2  813.51   309.4  830.47
#Mann= 7 ,-1 , 0
       0      .1       0    64.9    .045       0   66.04    .045       0
   83.46      .1       0  141.35    .016       0  200.92      .1       0
  230.71     .12       0
#XS Ineff= 2 , 0
                          119.29           792.7
Permanent Ineff=
       F       F
Bank Sta=66.04,83.46
XS Rating Curve= 0 ,0
Exp/Cntr=0.3,0.1

Type RM Length L Ch R = 1 ,1312.2  ,41.7,41.1,41.3
XS GIS Cut Line= 3
     1752927.102      362389.417     1753175.092      362353.114
     1753252.796      362299.833
#Sta/Elev= 30
       0  795.95   13.75796.1066    23.9  796.91    31.8  794.92    43.8  790.03
    55.7  789.29    59.7  787.61    63.6  784.47    71.6  780.18    79.6   777.4
    83.5  777.34    87.5  780.17    95.5  785.35   107.4  786.39   115.4   786.3
   139.2  782.66   167.1  781.57     191  781.96  222.71 780.655   234.7  781.21
  252.94788.2588   262.4  791.36   266.3  791.69   270.3  790.52   278.1  786.33
     282  785.89     286  787.31   301.7  798.94   317.4  805.61   344.8  834.32
#Mann= 6 ,-1 , 0
       0    .016       0   13.75      .1       0    71.6    .045       0
    87.5    .016       0  222.71      .1       0  252.94     .12       0
#XS Ineff= 2 , 0
                          107.64          786.68
Permanent Ineff=
       F       F
Bank Sta=71.6,87.5
XS Rating Curve= 0 ,0
Exp/Cntr=0.3,0.1

Type RM Length L Ch R = 1 ,1271.1  ,131.6,118.2,104.8
XS GIS Cut Line= 3
     1752935.088      362428.913     1753185.856      362394.694
      1753263.56      362341.413
#Sta/Elev= 30
       0  803.07    23.7  794.08    35.6  792.88    43.5  793.86   50.17 791.785
    63.3  788.57    75.1  775.94    79.1  775.22      87  773.37    94.9  775.94
    95.1776.0765   106.8   784.4   110.7  786.25   126.6  781.83   142.4  783.07
  184.53781.0372   213.6  780.99   229.4  779.18  244.15780.2213   249.1  781.14
   260.9  786.47   272.7  790.48  278.16790.6337   292.4  783.66   296.3  784.04
   300.2   786.4     308  793.97     312  796.78   327.7  803.56   347.3  818.76
#Mann= 8 ,-1 , 0
       0      .1       0   50.17    .016       0    79.1    .045       0
    94.9    .016       0    95.1      .1       0  184.53    .016       0
  244.15      .1       0  278.16     .12       0
#XS Ineff= 2 , 0
       0                   110.7       0
Permanent Ineff=
       F       F
Bank Sta=79.1,94.9
XS Rating Curve= 0 ,0
Exp/Cntr=0.3,0.1

Type RM Length L Ch R = 1 ,1152.9  ,253.3,253.5,253.7
XS GIS Cut Line= 3
     1753034.741         362554.     1753146.152      362459.494
     1753274.324      362377.611
#Sta/Elev= 30
       0  818.15    11.8  808.37    31.6   796.3    39.5  792.94    55.3  782.43
    71.1  772.99      79   770.8    82.9  770.97    88.8  773.45    98.7  778.85
   106.6  778.77   122.4  774.85   130.3  776.81   142.2  776.79   153.9  781.65
  160.65780.5715   196.8  778.75   208.5  779.96   212.4  781.23  215.51783.2874
  217.75784.6093   224.1  787.45   235.8  790.45   243.6  787.47   251.4  781.72
   255.3  780.32   259.2  781.29   274.8  795.09   282.6  799.47   298.2  805.03
#Mann= 6 ,-1 , 0
       0      .1       0    71.1    .045       0    88.8      .1       0
  160.65    .016       0  215.51      .1       0  217.75     .12       0
#XS Ineff= 2 , 0
                          102.25          779.28
Permanent Ineff=
       F       F
Bank Sta=71.1,88.8
XS Rating Curve= 0 ,0
Exp/Cntr=0.3,0.1

Type RM Length L Ch R = 1 ,899.4   ,292.7,304.1,314.8
XS GIS Cut Line= 2
     1753191.176      362752.444     1753352.635      362617.027
#Sta/Elev= 30
       0  831.19    8.45825.0961    15.9  819.59    19.9  816.95    35.8  807.56
    39.8   804.4    47.7  795.18    55.7   785.3    63.6  777.07    67.6  773.53
    71.6  771.02    74.7  769.48    75.5  769.08    79.5  768.39    89.7  768.91
    91.4  769.07    95.4  770.32   107.4  776.91   111.3  777.92   119.3  777.94
   123.3  777.12   127.2   775.8   131.2  775.57  174.25775.4567   178.9  775.28
   182.9   775.7   186.9  777.35   192.3778.8675   194.8  779.28   210.7  778.28
#Mann= 6 ,-1 , 0
       0     .12       0    8.45      .1       0    74.7    .045       0
    89.7      .1       0  174.25     .06       0   192.3    .016       0
Bank Sta=74.7,89.7
XS Rating Curve= 0 ,0
Exp/Cntr=0.3,0.1

Type RM Length L Ch R = 1 ,595.3   ,149.6,130,109.2
XS GIS Cut Line= 2
      1753244.29      362985.731     1753534.046      362928.306
#Sta/Elev= 30
       0  818.27       8  810.61    43.9  780.31    59.9  769.51    67.9  767.11
    95.8  767.51   105.8   765.8   115.8  765.62   120.8  765.71   127.7  766.73
   135.7  771.07   139.7  772.19   143.7  771.89   147.7  770.43   151.7  767.94
   155.7  767.06   167.7  766.08   183.6  771.04   199.6  781.07   203.6  782.26
   219.6   782.9   231.5  786.06   235.5  786.01   255.5  778.68  262.63775.1611
   275.4  770.23   279.4  769.48   283.4   769.6  292.74772.5253   295.4  773.31
#Mann= 5 ,-1 , 0
       0      .1       0   105.8    .045       0   120.8      .1       0
  262.63     .05       0  292.74     .06       0
#XS Ineff= 2 , 0
                          139.28          772.42
Permanent Ineff=
       F       F
Bank Sta=105.8,120.8
XS Rating Curve= 0 ,0
Exp/Cntr=0.3,0.1

Type RM Length L Ch R = 1 ,465.3   ,23.5,36.6,37.5
XS GIS Cut Line= 4
     1753246.402      363117.484     1753377.131       363108.89
     1753412.548      363045.609      1753551.35      363079.984
#Sta/Elev= 30
       0  814.72    19.8  798.01    43.7  783.51   48.87782.2001    51.6  781.62
    55.6  777.86    59.6  772.18    67.5  768.09    75.4  765.25   103.2  765.78
   115.1  765.22     131  767.36   142.5  765.56   153.9  764.76   165.4   764.3
   169.2  764.45   180.6   765.5   192.1  767.61   203.5  767.57   215.4  769.24
   227.4  769.49   239.3  767.77   243.2  768.66   251.2  772.06  265.16773.0515
   286.9  773.84   302.8  775.69  326.02773.7063   334.6  772.24   346.5  767.28
#Mann= 6 ,-1 , 0
       0     .12       0   48.87      .1       0   153.9    .045       0
   169.2      .1       0  265.16     .08       0  326.02     .12       0
#XS Ineff= 2 , 0
                          227.55          770.44
Permanent Ineff=
       F       F
Bank Sta=153.9,169.2
XS Rating Curve= 0 ,0
Exp/Cntr=0.3,0.1

Type RM Length L Ch R = 1 ,428.7   ,54.2,68.2,95.2
XS GIS Cut Line= 4
     1753250.568      363134.151     1753409.162      363123.734
     1753444.579      363060.453     1753550.568      363086.494
#Sta/Elev= 30
       0   808.5    15.9  800.58    27.8  791.92   44.69781.4442    51.6  774.55
    55.6  771.65    67.6  765.99    71.5  765.16    91.4   765.7   103.3  765.02
   119.2  767.61     147  768.04     151  767.12   158.9  763.43   166.6   762.9
   174.2  763.33   189.5  766.18   200.9  766.02     220  767.57   231.4   767.6
   235.4  768.35   243.2  771.67  260.08773.1841   282.1  774.02   289.9  775.72
   309.4  774.92  320.91773.4575     325  772.96   336.7  767.75   340.6  766.75
#Mann= 6 ,-1 , 0
       0     .12       0   44.69      .1       0   158.9    .045       0
   174.2      .1       0  260.08     .08       0  320.91     .12       0
#XS Ineff= 2 , 0
                          218.52          769.97
Permanent Ineff=
       F       F
Bank Sta=158.9,174.2
XS Rating Curve= 0 ,0
Exp/Cntr=0.3,0.1

Type RM Length L Ch R = 1 ,360.5   ,57.8,52.1,46.4
XS GIS Cut Line= 2
     1753252.796      363160.945      1753544.55      363192.068
#Sta/Elev= 30
       0  813.79    15.9  805.25    23.8  800.28    31.7  797.87   42.61792.2589
    51.5  785.36    59.5  780.58    63.4  777.52    71.4  769.89    75.3  767.03
    79.3  765.42    83.3  765.08    99.1  765.36     115  766.33   122.9  763.92
   138.8  763.67   146.7  762.78   154.6  762.52   162.6  762.89   174.5  764.98
   178.4  766.24  191.13772.7945   194.3  773.69   214.1  773.98  220.83  774.78
     230  774.87   241.9  773.95  250.53772.5861   265.6  771.14   293.4  765.92
#Mann= 7 ,-1 , 0
       0     .12       0   42.61      .1       0   146.7    .045       0
   162.6      .1       0  191.13     .12       0  220.83     .08       0
  250.53     .12       0
#XS Ineff= 2 , 0
                          224.49          775.82
Permanent Ineff=
       F       F
Bank Sta=146.7,162.6
XS Rating Curve= 0 ,0
Exp/Cntr=0.3,0.1

Type RM Length L Ch R = 1 ,308.4   ,135.9,101.5,52.5
XS GIS Cut Line= 3
     1753265.296       363247.75     1753434.837      363221.191
     1753555.401      363222.016
#Sta/Elev= 30
       0  821.88       4  819.33    31.9  808.47    43.9   805.1    47.9  802.59
    55.9  795.49   60.13791.2612    63.8  787.61    75.8  777.84    83.8  770.58
    87.8  768.61   107.8  767.94   111.8  767.23  121.98  762.56   127.7  761.32
   131.7  761.22   138.7  762.53  149.82763.9561   155.6  764.28   159.6  765.39
   167.6  769.32  179.62772.4749   206.6   774.6   222.2  773.86  238.69772.1945
   245.5  771.56   268.8  766.79   276.6  765.66   284.4  765.48   292.2  766.24
#Mann= 7 ,-1 , 0
       0     .12       0   60.13      .1       0  121.98    .045       0
   138.7      .1       0  149.82     .12       0  179.62     .08       0
  238.69     .12       0
#XS Ineff= 2 , 0
                          212.14          775.04
Permanent Ineff=
       F       F
Bank Sta=121.98,138.7
XS Rating Curve= 0 ,0
Exp/Cntr=0.3,0.1

Type RM Length L Ch R = 1 ,206.9   ,98.5,65.7,76.6
XS GIS Cut Line= 4
     1753301.957      363389.793     1753442.582      363366.355
     1753437.258      363235.905     1753561.824      363237.641
#Sta/Elev= 30
       0  816.04    31.7  799.13   53.01788.9869    63.4  783.12   82.95782.0237
     103  780.02   118.8  771.96   130.7  764.66   134.6  764.02   138.6  764.34
   142.6  765.94   162.4  767.12   178.2  766.58   182.1  766.06     194  761.39
   201.9  760.18   209.8  761.88   217.7  764.94   225.6  765.71   237.5  766.16
   249.4  764.56   265.2  765.97  278.71769.8936   304.3   774.7  337.79771.9597
     351  769.86   370.4   765.2   378.2  765.26   389.9  766.97   397.7  766.77
#Mann= 7 ,-1 , 0
       0     .12       0   53.01      .1       0   82.95     .12       0
     194    .045       0   209.8     .12       0  278.71     .08       0
  337.79     .12       0
#XS Ineff= 2 , 0
          165.94  769.22  232.82          768.72
Permanent Ineff=
       F       F
Bank Sta=194,209.8
XS Rating Curve= 0 ,0
Exp/Cntr=0.3,0.1
